HEC-RAS study LAURELCK.prj: LAURELCK

--- LAURELCK.g01 (geometry) --- (continued)

Type RM Length L Ch R = 1 ,16797.7 ,276.2,275,273.5
XS GIS Cut Line= 2
      2019929.47      273107.729     2019935.981      273496.184
#Sta/Elev= 30
       0  1809.2     9.8 1803.44      49 1782.12    81.6 1767.52   99.231762.006
   107.7 1761.42     111 1760.69   117.5 1756.93   120.8 1756.21   150.2 1755.77
   153.4 1755.24   156.7 1752.98     160 1749.62   163.2 1747.39     165 1747.21
   179.6    1747   182.8 1747.28   189.4 1749.93   192.6 1752.78   202.4 1754.75
   238.3 1754.61   244.9 1756.26  255.811757.338   274.2 1759.78   290.6 1760.49
   326.5 1763.44   352.6 1764.82  362.391766.168   375.4 1769.53   388.5  1774.4
#Mann= 6 ,-1 , 0
       0     .12       0   99.23    .016       0     165    .045       0
   182.8    .016       0  255.81     .08       0  362.39     .12       0
Bank Sta=165,182.8
XS Rating Curve= 0 ,0
Exp/Cntr=0.3,0.1

Type RM Length L Ch R = 1 ,16522.7 ,219.3,209,198.3
XS GIS Cut Line= 2
     2019646.267       273125.09     2019674.479      273483.163
#Sta/Elev= 30
       0 1757.54    1.761757.561   39.661757.519    68.6 1757.74    94.7 1755.61
   107.8 1755.23     111 1754.51  120.281749.029   127.4  1746.3   130.6 1745.65
   146.9 1744.44     160 1743.82   163.3 1744.36   166.7 1745.89   173.1 1749.29
  179.531750.026   189.4 1749.84   199.2 1748.66  209.16  1749.2   225.3    1749
   244.9 1749.96   267.8 1753.14  280.891756.607   297.1 1758.31   300.4 1760.36
   303.7  1761.3   310.2 1761.73   326.5 1767.72   339.6 1771.47   359.2 1776.11
#Mann= 9 ,-1 , 0
       0     .12       0    1.76     .06       0   39.66     .08       0
  120.28     .12       0   146.9    .045       0   166.7     .08       0
  179.53    .016       0  209.16     .08       0  280.89     .12       0
Bank Sta=146.9,166.7
XS Rating Curve= 0 ,0
Exp/Cntr=0.3,0.1

Type RM Length L Ch R = 1 ,16313.8 ,49.2,52.5,55.9
XS GIS Cut Line= 5
     2019362.383      273082.233      2019379.31       273136.92
     2019435.764       273285.68     2019519.314      273423.484
     2019560.547      273515.715
#Sta/Elev= 30
       0 1765.27   15.771761.941      35 1758.73    50.9 1757.05      80 1757.18
  191.211751.282   206.6  1750.8   216.4 1749.75   229.2 1746.55   238.9 1742.34
  241.36  1741.8   261.5 1741.51   264.7 1741.76   274.4 1746.05   303.4 1746.32
   319.5 1745.95   325.9 1744.98  328.171745.386   332.4 1746.15   351.7  1746.4
   364.6 1748.59   367.8 1749.82   371.1 1752.07   374.3 1755.52   380.8 1764.12
     384 1766.66   387.3 1767.59  408.481768.946   436.2 1770.09   478.5 1774.79
#Mann= 7 ,-1 , 0
       0     .12       0   15.77    .016       0  191.21     .08       0
  241.36    .045       0   264.7    .016       0  328.17     .12       0
  408.48     .06       0
#XS Ineff= 2 , 0
                          276.99         1748.83
Permanent Ineff=
       F       F
Bank Sta=241.36,264.7
XS Rating Curve= 0 ,0
Exp/Cntr=0.3,0.1

Type RM Length L Ch R = 1 ,16261.2 ,216.8,217.6,218.3
XS GIS Cut Line= 4
     2019305.091       273099.16     2019348.696      273202.489
     2019442.274      273419.144     2019523.654      273527.651
#Sta/Elev= 30
       0 1780.56   15.451778.443    38.4 1770.94    67.3 1762.41    86.5 1758.45
   125.3 1753.65   194.1 1751.56   210.5 1750.27  221.931748.652  225.991748.344
   246.5 1748.22   249.8 1747.08   256.4 1742.61   258.4 1742.05   279.3 1741.56
   282.6  1741.8   289.2 1744.75   292.4 1745.19  297.261744.276   312.1 1744.09
   328.5 1746.21  347.731746.623   351.4 1747.77   354.6 1749.57   361.1 1754.27
     374  1766.9   377.2  1768.6   380.4 1769.44  464.331775.638   483.8 1776.87
#Mann= 9 ,-1 , 0
       0     .12       0   15.45     .08       0  221.93     .06       0
  225.99    .016       0   258.4    .045       0   282.6     .08       0
  297.26    .016       0  347.73     .12       0  464.33     .06       0
#XS Ineff= 2 , 0
                          303.98         1749.36
Permanent Ineff=
       F       F
Bank Sta=258.4,282.6
XS Rating Curve= 0 ,0
Exp/Cntr=0.3,0.1

Type RM Length L Ch R = 1 ,16043.7 ,145.7,149.2,151.9
XS GIS Cut Line= 3
     2019185.113      273261.809     2019197.048      273365.976
      2019304.47      273650.264
#Sta/Elev= 30
       0    1770    16.4 1768.03    22.9 1768.18    62.2 1765.03    78.6 1760.49
    98.3 1751.16   114.6 1745.39   137.5 1741.45  148.751741.786   196.4 1741.56
   206.2 1737.58   212.7 1737.24   222.5 1737.42     225 1738.02  236.131743.768
   238.8 1745.32   242.1 1746.16  283.611747.329   304.2 1747.23   307.4 1747.76
  317.851754.901   327.1 1759.85  350.551775.905   356.5 1778.35   359.7    1779
   376.1 1778.39   379.3 1779.23     3861783.646   392.4 1787.43   408.8 1791.87
#Mann= 9 ,-1 , 0
       0     .06       0  148.75     .12       0   206.2    .045       0
     225     .12       0  236.13     .08       0  283.61    .016       0
  317.85     .12       0  350.55    .016       0     386     .06       0
#XS Ineff= 2 , 0
          185.37 1749.17
Permanent Ineff=
       F       F
Bank Sta=206.2,225
XS Rating Curve= 0 ,0
Exp/Cntr=0.3,0.1

Type RM Length L Ch R = 1 ,15894.5 ,119.5,119.6,118.6
XS GIS Cut Line= 3
     2019106.988      273284.595     2019083.116      273414.804
     2019151.476      273728.389
#Sta/Elev= 30
       0 1770.18    74.3 1762.95   100.1 1759.52   111.71756.954   125.9 1752.68
   132.4 1751.73   135.6 1750.15   138.9 1746.66   142.2 1741.38   145.5 1738.31
   155.3 1736.29   161.8 1734.12   171.7  1733.2   178.2 1734.71     188 1737.18
   201.2 1738.82   289.6 1741.98  321.351745.599   338.7 1745.37   345.2 1746.54
  351.581749.028   364.9 1757.12   368.2 1758.49   374.7 1759.72   384.6 1759.48
   387.8 1760.34  390.77  1762.5   400.9 1772.69   404.2 1775.36   453.3 1809.14
#Mann= 7 ,-1 , 0
       0     .06       0   111.7     .12       0   161.8    .045       0
   178.2     .12       0  321.35    .016       0  351.58     .08       0
  390.77     .12       0
Bank Sta=161.8,178.2
XS Rating Curve= 0 ,0
Exp/Cntr=0.3,0.1

Type RM Length L Ch R = 1 ,15774.9 ,176.6,181.7,186.7
XS GIS Cut Line= 3
     2018996.311      273325.828     2018955.078      273384.422
     2019052.734      273771.791
#Sta/Elev= 30
       0 1760.34    52.1 1756.27    71.6 1752.04  108.871747.904   127.3 1746.87
   133.9 1745.77   156.8 1732.11   163.3 1731.48   173.2 1731.49   177.1 1732.16
   186.3 1735.57   209.2 1736.28  232.47 1738.29   287.8  1737.8   300.9 1738.49
  305.641740.398     314 1745.95   317.2 1746.86   343.4  1747.9   346.7  1749.1
  354.311756.667   359.8 1762.12   366.4 1767.03   382.7 1780.99   399.1 1793.88
   405.6 1798.08   415.5 1802.66   431.8 1813.16   464.6 1830.48   471.1 1834.48
#Mann= 7 ,-1 , 0
       0     .08       0  108.87     .12       0   156.8    .045       0
   177.1     .12       0  232.47     .08       0  305.64    .016       0
  354.31     .12       0
Bank Sta=156.8,177.1
XS Rating Curve= 0 ,0
Exp/Cntr=0.3,0.1

Type RM Length L Ch R = 1 ,15593.2 ,207.5,206.9,207.6
XS GIS Cut Line= 2
     2018807.509      273303.041     2018818.359      273778.302
#Sta/Elev= 30
       0 1749.55    13.1 1745.07    26.2 1744.23    39.3 1740.48    60.11739.293
    95.1 1740.36  159.481739.992   190.2 1740.27  193.921739.121   203.3 1734.07
   239.3 1729.39   245.9 1728.76   257.7 1729.53   265.6 1730.14   268.8  1731.3
     282 1737.02  291.66 1743.38   298.3 1747.95   301.6 1749.23  326.011750.038
   334.4 1751.21   350.8 1757.51   357.4 1761.28   360.6 1764.83   370.5 1792.69
  374.141798.502   383.6 1809.31   390.1 1815.65   403.3 1826.17   475.4 1869.55
#Mann= 9 ,-1 , 0
       0    .016       0    60.1     .08       0  159.48    .016       0
  193.92     .12       0   239.3    .045       0   257.7     .12       0
  291.66    .016       0  326.01     .08       0  374.14     .12       0
#XS Ineff= 2 , 0
          218.75 1744.87
Permanent Ineff=
       F       F
Bank Sta=239.3,257.7
XS Rating Curve= 0 ,0
Exp/Cntr=0.3,0.1

Type RM Length L Ch R = 1 ,15386.3 ,204.7,202.6,198.4
XS GIS Cut Line= 2
     2018605.686      273320.403     2018611.111      273759.856
#Sta/Elev= 30
       0 1739.43    29.5 1736.22   137.8 1733.72  160.891731.738   173.8 1729.14
  185.841730.794   196.8 1731.96   206.6 1728.79   213.2 1728.75   216.5 1727.73
   219.7 1726.42   236.1 1726.08   239.4 1726.43  240.62 1727.57   245.31732.917
   249.3 1738.23   252.5 1741.29   259.1 1744.26   265.7 1744.47   268.9 1745.56
   278.8 1755.26   282.1 1756.64   291.9 1756.71  308.591754.959   311.6 1756.19
   314.9 1761.36   321.4 1778.63   324.7 1782.63  338.131792.099   439.5  1852.2
#Mann= 8 ,-1 , 0
       0     .06       0  160.89    .016       0  185.84     .12       0
   216.5    .045       0  240.62     .12       0   245.3    .016       0
  308.59     .08       0  338.13     .12       0
#XS Ineff= 2 , 0
          196.02 1742.65
Permanent Ineff=
       F       F
Bank Sta=216.5,240.62
XS Rating Curve= 0 ,0
Exp/Cntr=0.3,0.1

Type RM Length L Ch R = 1 ,15183.6 ,33.4,33,33.4
XS GIS Cut Line= 3
     2018388.672      273234.682     2018436.415      273655.689
     2018492.838      273780.472
#Sta/Elev= 30
       0 1751.47      181737.984    26.1 1732.83    32.6 1730.64   69.81 1729.28
  156.791729.024  197.251729.532   221.6 1729.35   231.4 1725.32     251 1724.16
   257.5 1725.82     264  1728.5  269.861727.706   277.91727.375  304.591728.237
   329.2 1729.89   384.6 1737.55  426.791746.588   443.3 1751.53  453.321758.459
   459.6 1761.81   485.7 1761.39   488.9 1762.63   492.2 1765.01   495.4 1769.52
  498.641776.786     502 1784.11   505.2 1787.49   531.3 1806.48   560.6 1824.56
#Mann= 13 ,-1 , 0
       0    .016       0      18     .12       0   69.81     .08       0
  156.79     .06       0  197.25    .016       0   231.4    .045       0
   257.5    .016       0  269.86     .12       0   277.9    .016       0
  304.59     .08       0  426.79     .12       0  453.32    .016       0
  498.64     .12       0
Bank Sta=231.4,257.5
XS Rating Curve= 0 ,0
Exp/Cntr=0.3,0.1

Type RM Length L Ch R = 1 ,15150.7 ,114.6,114.6,114.9
XS GIS Cut Line= 3
     2018359.375      273237.937     2018407.118      273658.944
     2018463.542      273783.727
#Sta/Elev= 30
       0 1746.56   13.441737.664    19.6 1734.63    26.1 1733.17   72.121729.322
   140.2 1728.35  203.991729.489   211.8 1728.76   221.6 1723.72   231.4 1723.37
   241.2 1723.95   257.5 1729.22   273.8 1727.07   322.7 1728.68   410.7 1736.47
   446.5  1744.7  452.73 1747.58  455.641748.686   462.8 1751.91   472.6 1759.85
   475.9 1761.48   498.7 1761.55     502 1762.46   505.2 1764.57   508.5 1768.73
  510.751773.694   518.3 1788.83   521.5 1792.42   547.6 1811.44   560.6 1819.26
#Mann= 9 ,-1 , 0
       0    .016       0   13.44     .12       0   72.12     .06       0
  203.99    .016       0   221.6    .045       0   241.2    .016       0
  452.73     .12       0  455.64    .016       0  510.75     .12       0
Bank Sta=221.6,241.2
XS Rating Curve= 0 ,0
Exp/Cntr=0.3,0.1

Type RM Length L Ch R = 1 ,15036.1 ,384.1,373.4,362.3
XS GIS Cut Line= 4
     2018180.338      273267.234     2018263.889      273371.401
     2018305.121      273674.135     2018390.842      273835.811
#Sta/Elev= 30
       0 1766.84     6.5 1763.18    29.3 1745.95    45.6 1738.46    58.6 1735.13
   95.461732.317   149.8 1728.85  166.051726.191   195.3 1723.02     205 1722.02
   213.4 1723.21     2271725.242  276.641726.289   331.8    1725   361.1 1728.09
  423.281729.279   452.1  1731.1  475.941734.088   494.6 1742.22     511 1743.14
   514.2 1744.38   537.1 1760.45   546.9 1762.35   563.2 1762.61  567.651765.665
   569.8 1768.44   579.6 1785.45   582.8 1789.05   612.2 1810.91   622.1  1816.7
#Mann= 10 ,-1 , 0
       0     .12       0   95.46     .06       0  166.05     .12       0
   195.3    .045       0   213.4     .12       0     227    .016       0
  276.64     .06       0  423.28     .12       0  475.94    .016       0
  567.65     .12       0
#XS Ineff= 2 , 0
                          322.16         1731.59
Permanent Ineff=
       F       F
Bank Sta=195.3,213.4
XS Rating Curve= 0 ,0
Exp/Cntr=0.3,0.1

Type RM Length L Ch R = 1 ,14662.6 ,198,212.1,225.2
XS GIS Cut Line= 2
     2017903.646       273441.93     2018213.976      273870.533
#Sta/Elev= 30
       0 1758.42    29.4 1742.02    45.7 1730.08    55.5 1719.55    68.6 1717.53
    75.1 1716.96    86.5 1717.31   99.631719.993   107.8 1723.09  123.39 1722.02
     147 1724.03  177.411722.927   202.5 1721.73  244.411721.727  296.451720.844
   316.8 1719.34   333.2 1721.21   388.7 1722.32   399.91723.948   408.3 1727.04
   427.9 1727.06   447.5 1728.57  457.781733.208   467.1 1742.48   483.4 1744.52
   486.7 1747.52   493.2 1755.69     503 1765.08   509.6 1766.73   529.2 1766.62
#Mann= 10 ,-1 , 0
       0     .12       0    68.6    .045       0    86.5     .12       0
   99.63    .016       0  123.39     .12       0  177.41     .06       0
  244.41     .12       0  296.45     .06       0   399.9     .12       0
  457.78    .016       0
#XS Ineff= 2 , 0
                          361.36         1725.44
Permanent Ineff=
       F       F
Bank Sta=68.6,86.5
XS Rating Curve= 0 ,0
Exp/Cntr=0.3,0.1

Type RM Length L Ch R = 1 ,14450.6 ,202.7,203.4,204.1
XS GIS Cut Line= 2
     2017775.143      273488.483     2017786.024      273990.541
#Sta/Elev= 30
       0 1756.72    19.6  1748.7    39.1 1741.69    78.3 1719.49    84.8    1718
   101.1 1716.33   107.6 1714.06   117.4 1713.22   127.2    1713   135.4 1713.32
   140.2 1714.97   146.7 1718.57  156.451716.819  189.361716.442   215.2  1716.7
     287 1713.92  296.291714.815   309.21715.093   329.4 1715.52   355.4 1718.81
   378.3 1719.48   394.6 1721.14   401.1 1722.43   417.4 1727.63   430.4    1734
   446.7 1740.83   466.3 1745.92   485.9 1749.68   492.4 1752.05   502.2 1757.06
#Mann= 7 ,-1 , 0
       0     .12       0   117.4    .045       0   135.4     .12       0
  156.45    .016       0  189.36     .12       0  296.29     .06       0
   309.2     .12       0
Bank Sta=117.4,135.4
XS Rating Curve= 0 ,0
Exp/Cntr=0.3,0.1

Type RM Length L Ch R = 1 ,14247.2 ,175.9,176.1,176.2
XS GIS Cut Line= 3
     2017582.435      273472.858     2017575.925      273876.503
     2017557.509      273980.125
#Sta/Elev= 30
       0 1762.71      13 1752.27    42.3 1732.87    65.1 1722.16    84.6 1708.99
    87.9 1707.88   100.9 1707.48   105.6 1708.09   123.7 1713.85     127 1713.62
   130.81712.518   143.2 1711.86  163.861712.847   211.6 1712.85   237.7 1711.63
   250.7 1712.54     280 1711.22   309.3 1711.78   322.3 1711.28   332.1 1711.94
   338.6 1711.16   354.9 1713.32   390.7  1715.2   397.2  1716.8   406.9 1721.58
   413.3 1723.73   435.6 1728.66   451.5 1733.91   473.9    1739   508.9 1750.09
#Mann= 5 ,-1 , 0
       0     .12       0    87.9    .045       0   105.6     .12       0
   130.8    .016       0  163.86     .12       0
Bank Sta=87.9,105.6
XS Rating Curve= 0 ,0
Exp/Cntr=0.3,0.1

Type RM Length L Ch R = 1 ,14071.1 ,155.9,159.4,162.2
XS GIS Cut Line= 3
     2017409.939      273485.333     2017407.769      273851.002
     2017405.599      273946.488
#Sta/Elev= 30
       0 1770.02    19.6 1758.66    29.4 1751.54    32.6 1748.78    42.4 1737.61
    55.5 1727.06    71.8 1717.04    78.4 1713.61    84.9 1708.18    91.4 1705.61
    94.7 1705.23   104.5 1704.65   109.7 1705.54   117.5 1707.51  123.52 1707.71
   143.7 1707.33   156.7  1709.4  173.151709.045   189.4 1708.15   205.7 1708.95
   231.8  1707.7   248.1 1707.59   279.41708.508   287.3 1707.45   293.8 1708.47
   303.6 1711.27     333  1716.2     388 1723.65   403.9 1728.16   461.2 1750.66
#Mann= 6 ,-1 , 0
       0     .12       0    94.7    .045       0   109.7     .12       0
  123.52    .016       0  173.15     .06       0   279.4     .12       0
Bank Sta=94.7,109.7
XS Rating Curve= 0 ,0
Exp/Cntr=0.3,0.1

Type RM Length L Ch R = 1 ,13911.7 ,56.6,56.2,56.8
XS GIS Cut Line= 4
     2017282.552      273461.462     2017272.786      273636.158
     2017279.297      273810.854     2017321.614      273921.531
#Sta/Elev= 30
       0  1789.1     6.5 1785.63     9.7 1783.27    51.8  1765.4      68  1757.9
    77.8 1752.58    87.5 1749.13    97.2 1743.46   123.1 1731.43   132.8 1725.11
   152.3  1717.6     162 1712.32   165.2 1711.53   181.4 1710.32   184.7 1709.47
  192.621704.755   199.7 1702.29   204.1 1701.84   214.7 1702.06   236.5 1705.05
  256.421703.955   278.6 1704.15  285.981705.575   301.2 1707.65  334.761709.129
   375.4 1710.78   378.6 1711.42   394.6 1717.21   423.4 1729.85   468.3 1740.48
#Mann= 7 ,-1 , 0
       0     .12       0  192.62    .016       0   199.7    .045       0
   214.7    .016       0  256.42     .08       0  285.98     .06       0
  334.76     .12       0
Bank Sta=199.7,214.7
XS Rating Curve= 0 ,0
Exp/Cntr=0.3,0.1

Type RM Length L Ch R = 1 ,13855.5 ,88.2,65.7,42.1
XS GIS Cut Line= 3
     2017235.243      273461.462     2017233.073      273778.302
     2017298.177      273928.041
#Sta/Elev= 30
       0 1787.68    35.9 1769.07    75.1 1750.39   107.8 1736.88   120.9 1730.19
   133.9 1726.48   140.5 1722.83   150.3 1714.95   160.1 1708.18   166.6 1706.44
  201.121706.064   215.6 1706.13   225.4  1704.5   231.9 1702.08   241.7 1701.13
   261.3 1701.47     2681701.464  285.641702.827     294 1705.17     307 1707.08
   326.6 1707.82  346.181709.609  355.391710.516   378.9 1712.81   388.7 1714.51
   398.5 1718.04   411.6 1721.66   450.7 1730.37   463.8 1732.58   480.1 1737.22
#Mann= 8 ,-1 , 0
       0     .12       0  201.12    .016       0   231.9    .045       0
   261.3    .016       0     268     .08       0  285.64     .12       0
  346.18     .06       0  355.39     .12       0
Bank Sta=231.9,261.3
XS Rating Curve= 0 ,0
Exp/Cntr=0.3,0.1

Type RM Length L Ch R = 1 ,13789.9 ,42.8,42.7,42.6
XS GIS Cut Line= 4
     2017036.675      273464.717     2017009.548      273599.265
     2017223.307      273784.812      2017275.39      273952.998
#Sta/Elev= 30
       0 1788.46      36 1767.78      49 1761.43   107.8 1739.57   117.6 1732.78
   120.9 1731.58   130.7 1731.16     147 1726.78     160 1724.77   195.8 1709.12
   208.8 1706.66   218.6 1701.99  272.651702.932  302.981703.371   332.5 1704.34
   348.7 1706.39     352 1705.67   358.5 1701.81  361.591700.902  362.771700.804
   371.5 1700.67   382.1 1700.85   387.8 1702.05   397.5 1706.14   452.9 1709.77
     492 1715.67   560.5 1729.84   576.8 1735.04   593.1 1738.75   596.4 1740.42
#Mann= 6 ,-1 , 0
       0     .12       0  272.65     .06       0  302.98    .016       0
  361.59     .08       0  362.77    .045       0   382.1     .12       0
#XS Ineff= 2 , 0
          296.59 1711.34
Permanent Ineff=
       F       F
Bank Sta=362.77,382.1
XS Rating Curve= 0 ,0
Exp/Cntr=0.3,0.1

Type RM Length L Ch R = 1 ,13747.2 ,195.8,200.6,205.4
XS GIS Cut Line= 4
      2017006.51      273459.074      2016975.26      273627.477
     2017211.371      273830.602     2017249.566      273969.491
#Sta/Elev= 30
       0 1792.97    19.4 1782.15      42 1768.52    54.9 1761.45    67.9  1755.3
      84  1751.1      97 1744.49   113.1 1738.88   129.3  1738.1   135.7    1736
   148.7 1729.15   177.8    1712   194.2 1704.06   207.3 1702.15   213.9  1701.9
   264.11702.737   338.5 1703.96  354.691703.451   387.7 1705.89  405.46 1700.38
   420.4 1700.14     427 1700.31   430.3 1700.89   440.1 1704.45   476.2 1708.46
   489.3 1710.74   505.7 1715.09   574.4  1726.9   607.1 1740.67   626.8 1751.32
#Mann= 5 ,-1 , 0
       0     .12       0   264.1    .016       0  354.69     .12       0
  405.46    .045       0     427     .12       0
#XS Ineff= 2 , 0
          325.14 1713.38
Permanent Ineff=
       F       F
Bank Sta=405.46,427
XS Rating Curve= 0 ,0
Exp/Cntr=0.3,0.1

Type RM Length L Ch R = 1 ,13546.6 ,377.6,383.7,389.3
XS GIS Cut Line= 3
     2016822.018       273668.17     2017044.675      273962.441
      2017073.32       274074.42
#Sta/Elev= 30
       0 1723.21     3.3 1720.92     6.5 1719.84    16.3 1718.84    26.1 1712.31
    39.2 1706.86      49  1704.4    68.6  1703.8    91.4 1701.54   114.3 1702.07
   166.6 1700.94   225.3 1701.37   248.11700.579  284.171700.955   300.4  1700.6
  304.651699.815   309.9 1698.46   316.8 1696.79     320 1696.75   326.6 1696.96
   333.1 1698.65     356 1710.23   378.6 1724.81   388.3 1732.13   417.2 1757.16
   420.4 1760.86     430 1769.26   436.4 1777.09   462.1 1801.01   484.6 1819.65
#Mann= 6 ,-1 , 0
       0     .12       0   248.1     .06       0  284.17     .12       0
  304.65     .08       0   309.9    .045       0   333.1     .12       0
#XS Ineff= 2 , 0
          221.59  1716.2
Permanent Ineff=
       F       F
Bank Sta=309.9,333.1
XS Rating Curve= 0 ,0
Exp/Cntr=0.3,0.1

Type RM Length L Ch R = 1 ,13162.9 ,340.4,342.3,343.4
XS GIS Cut Line= 3
     2016700.087      273818.015     2016674.045      273989.456
     2016784.722      274243.363
#Sta/Elev= 30
       0 1740.38    32.7 1737.33   121.1 1725.39   127.6  1723.5   140.7  1715.6
   147.2 1713.96   170.1 1702.47   183.2 1697.31     193 1695.77  223.621694.098
   235.3 1690.33   251.6 1688.66   261.2  1690.2   271.2 1689.68   277.7 1691.03
   287.5 1691.57     294 1694.65   297.2 1699.96     307 1727.07   310.3 1734.54
   313.5 1739.81     320 1747.39   365.7  1780.6   391.7 1802.87  396.771805.042
   404.8 1806.15   421.1 1806.15  433.631814.095   443.9 1829.81   450.4 1835.78
#Mann= 6 ,-1 , 0
       0     .12       0  223.62     .08       0   261.2    .045       0
   277.7     .12       0  396.77    .016       0  433.63     .12       0
Bank Sta=261.2,277.7
XS Rating Curve= 0 ,0
Exp/Cntr=0.3,0.1

Type RM Length L Ch R = 1 ,12820.6 ,324,321,318.5
XS GIS Cut Line= 3
     2016363.715      273833.206     2016346.354      273993.797
     2016459.201      274323.658
#Sta/Elev= 30
       0 1750.08    77.5 1736.21   100.2 1731.47   113.1 1730.08     126 1727.26
  144.071725.302     168 1722.25   171.3 1720.84   174.6 1718.18   177.8 1714.58
   200.6 1692.61   207.1 1686.89   216.9 1679.72   220.2 1678.06   223.4 1677.49
   239.7 1675.67   246.2 1674.95     262 1675.88   278.8 1679.45   308.2 1681.35
   314.7 1682.73   324.4 1688.84   334.2 1692.04   337.5 1693.86   347.2 1701.57
   353.8 1703.25   392.9 1709.71   418.9 1717.26   487.4 1745.84   510.2 1756.83
#Mann= 4 ,-1 , 0
       0     .06       0  144.07     .12       0   239.7    .045       0
     262     .12       0
Bank Sta=239.7,262
XS Rating Curve= 0 ,0
Exp/Cntr=0.3,0.1

Type RM Length L Ch R = 1 ,12499.6 ,262.8,259.9,257.1
XS GIS Cut Line= 3
     2016046.875      273948.224     2016027.344      274087.113
     2016153.212      274341.019
#Sta/Elev= 30
       0 1734.42    16.3 1729.99   62.291720.629   101.1 1715.21  123.951713.352
     137 1712.87   146.8 1709.56   156.5 1707.86   163.1 1706.05   172.8 1700.73
   195.6 1684.26   205.4 1678.36   215.2 1673.66  222.28  1672.5     225 1672.22
   234.7 1672.08     251 1672.23  255.251672.511     264 1673.68   273.8  1674.1
   283.6  1675.5   290.1 1677.25   303.1 1683.38   319.4 1687.78   329.71689.747
   361.8 1695.96  389.731703.228   397.6 1705.89   410.6 1711.26   423.6 1717.76
#Mann= 9 ,-1 , 0
       0     .12       0   62.29     .06       0  123.95     .12       0
  222.28     .08       0     225    .045       0     251     .08       0
  255.25     .12       0   329.7     .06       0  389.73     .12       0
Bank Sta=225,251
XS Rating Curve= 0 ,0
Exp/Cntr=0.3,0.1

Type RM Length L Ch R = 1 ,12239.7 ,117.6,115,112.4
XS GIS Cut Line= 3
     2015766.927      274071.922     2015749.566      274156.557
     2015940.538      274443.015
#Sta/Elev= 30
       0 1718.91    22.4 1709.71      32 1706.49      64 1697.92    86.4 1689.95
    99.5 1686.57   112.6 1685.46  160.611685.892  162.261685.857   204.4 1684.67
   207.7 1684.15  212.891681.786  233.261668.656   237.2 1667.61   260.2 1667.48
   263.5 1667.56  266.14 1668.08  267.871668.633     293 1677.48  304.261678.055
   319.2 1680.13   332.3  1680.6   345.4 1682.16   355.3 1683.78   365.1 1687.73
   371.7 1691.12   381.5 1697.66     411 1721.13   420.8  1726.9   430.7 1734.42
#Mann= 10 ,-1 , 0
       0     .12       0  160.61     .06       0  162.26     .08       0
  212.89     .12       0  233.26     .08       0   237.2    .045       0
   263.5     .08       0  266.14     .12       0  267.87     .08       0
  304.26     .12       0
Bank Sta=237.2,263.5
XS Rating Curve= 0 ,0
Exp/Cntr=0.3,0.1

Type RM Length L Ch R = 1 ,12124.7 ,37.9,37.9,37.9
XS GIS Cut Line= 2
     2015593.316      274178.258     2015836.371      274464.717
#Sta/Elev= 30
       0  1700.6    26.1 1689.35    45.7 1684.59    55.5 1682.93    81.7 1680.93
   101.3 1680.63  121.691681.197  170.531682.172   202.5 1679.52   205.8 1678.11
  209.271675.564   212.3 1672.79  218.341668.997   222.1 1667.53   227.1 1666.71
   241.7 1666.38   254.8 1666.71   264.6  1669.4   271.1 1672.52   274.4 1673.42
  282.63 1673.77   290.7 1673.67     294 1674.26   300.5 1678.98   303.8 1680.65
   316.9 1685.11   339.7 1695.77   346.3 1699.49   362.6 1710.42   375.7 1720.31
#Mann= 8 ,-1 , 0
       0     .12       0  121.69     .08       0  170.53     .06       0
  209.27    .016       0  218.34     .08       0   227.1    .045       0
   254.8     .08       0  282.63     .12       0
Bank Sta=227.1,254.8
XS Rating Curve= 0 ,0
Exp/Cntr=0.3,0.1

Type RM Length L Ch R = 1 ,12086.8 ,291.5,304.8,317.8
XS GIS Cut Line= 2
     2015558.594       274195.62     2015801.649      274482.078
#Sta/Elev= 30
       0 1702.69    16.3 1693.25    26.1 1688.88    32.7 1686.61    52.3  1681.5
    65.3 1679.86    78.4  1679.2   129.71679.644     147 1679.85   173.1 1677.81
   202.5  1677.3   205.8 1676.84   209.1 1675.49   215.6 1670.25   218.9 1668.93
   225.4 1666.87   232.9  1666.1   235.2 1666.01   264.6 1666.25   267.9 1666.56
   271.1 1667.72   280.9 1672.47  294.261673.085   300.5 1673.28   303.8    1675
   310.3 1679.74   316.9 1682.33   336.5 1692.09   346.3 1698.55   375.7 1720.26
#Mann= 5 ,-1 , 0
       0     .12       0   129.7    .016       0   232.9    .045       0
   264.6    .016       0  294.26     .12       0
Bank Sta=232.9,264.6
XS Rating Curve= 0 ,0
Exp/Cntr=0.3,0.1

Type RM Length L Ch R = 1 ,11782.1 ,290.3,292.7,294.5
XS GIS Cut Line= 3
     2015400.173      274239.022     2015447.917      274631.818
      2015497.83      274696.922
#Sta/Elev= 30
       0 1707.09      36 1689.58    81.8  1673.2   104.6 1671.26   150.4  1671.2
   153.7  1670.7   166.8 1664.24   173.3 1662.59   196.2 1663.11   199.5 1662.53
   209.3 1657.67   231.6 1656.28   238.7  1656.1   246.6 1656.75   274.7 1658.69
   281.2 1660.34     291 1666.36   307.4 1680.93   320.5  1690.5   336.8 1696.38
  372.461706.856   382.6 1709.27   408.3 1712.64   424.1 1712.12   427.2 1712.64
  432.351715.566   436.7 1718.98     443 1721.62     462 1724.55   477.7 1728.24
#Mann= 5 ,-1 , 0
       0     .12       0   231.6    .045       0   246.6     .12       0
  372.46    .016       0  432.35     .12       0
Bank Sta=231.6,246.6
XS Rating Curve= 0 ,0
Exp/Cntr=0.3,0.1

Type RM Length L Ch R = 1 ,11489.4 ,434.7,421.1,407.2
XS GIS Cut Line= 3
     2015135.417      274271.574     2015144.097      274627.477
     2015230.903      274714.283
#Sta/Elev= 30
       0 1738.42    22.9 1719.86    39.2 1707.77    71.8 1685.06    94.7 1672.94
     111 1659.39   120.8  1655.5   130.6 1653.95   137.2 1653.78   156.8 1655.37
   163.3 1651.93   166.6 1650.93   186.2 1650.61     196 1651.02     209 1655.22
   218.8 1661.77   225.4 1664.86   248.2 1665.98  283.511668.502  290.391669.234
   320.1 1671.52  349.08 1675.57   352.7 1676.62   362.5 1681.94   378.6 1687.17
  384.791688.254   414.2 1691.75  447.641697.832   456.2 1699.08   478.8 1699.27
#Mann= 9 ,-1 , 0
       0     .12       0   166.6    .045       0     196     .12       0
   248.2     .08       0  283.51     .06       0  290.39     .08       0
  349.08     .12       0  384.79     .06       0  447.64    .016       0
Bank Sta=166.6,196
XS Rating Curve= 0 ,0
Exp/Cntr=0.3,0.1

Type RM Length L Ch R = 1 ,11068.2 ,441.2,457,472.1
XS GIS Cut Line= 3
     2014699.219      274349.699     2014705.729      274464.717
     2014924.913      274749.005
#Sta/Elev= 30
       0 1718.46    25.6 1708.46   115.2 1684.22     125 1682.81   131.5 1680.49
   144.6  1677.9   151.1 1675.96   157.6 1672.45   164.2 1665.97   167.4 1663.33
   173.9 1659.26   183.7 1650.41     187  1648.4   190.3 1647.25   193.5 1647.05
   216.4 1646.75     220 1646.84     236 1649.09   252.3 1649.57   265.3  1651.8
  278.771652.172   304.5 1653.37   353.4 1658.05   392.6 1660.84  439.831666.746
   448.1 1668.32   454.6 1670.85   461.1 1674.64   470.9 1681.82   474.2 1683.63
#Mann= 5 ,-1 , 0
       0     .12       0   193.5    .045       0     220     .12       0
  278.77     .06       0  439.83     .12       0
Bank Sta=193.5,220
XS Rating Curve= 0 ,0
Exp/Cntr=0.3,0.1

Type RM Length L Ch R = 1 ,10611.2 ,288.5,288.3,288.2
XS GIS Cut Line= 2
     2014411.862      274405.149     2014387.123      274897.337
#Sta/Elev= 30
       0 1700.26    71.8 1673.78    88.1 1664.96   107.7 1652.52   114.2 1649.28
   133.8 1647.16  163.04    1647  222.371648.216   228.4 1647.77   241.5 1641.98
     248 1641.03   287.2 1642.17   336.2 1639.49   349.2 1639.14     359  1639.7
   362.3 1643.45     372  1664.9   381.8 1675.13   385.1 1678.29   391.6 1682.59
   401.4  1686.7     408 1690.92  413.831692.952     421 1693.76  439.821693.809
   443.8 1693.36   447.1 1694.98   456.9    1704   463.4 1708.08   492.8 1718.66
#Mann= 7 ,-1 , 0
       0     .12       0  163.04     .06       0  222.37     .12       0
   336.2    .045       0     359     .12       0  413.83    .016       0
  439.82     .12       0
Bank Sta=336.2,359
XS Rating Curve= 0 ,0
Exp/Cntr=0.3,0.1

Type RM Length L Ch R = 1 ,10322.9 ,395.9,394.9,393.2
XS GIS Cut Line= 2
     2014126.302      274425.654      2014100.26      274887.894
#Sta/Elev= 30
       0 1672.18    52.2 1650.98      62 1647.92    78.2 1645.32   107.6 1642.44
   146.7 1643.44   169.5 1643.02   189.1 1640.51   202.1 1635.94   228.2 1637.16
   257.6 1637.25   281.6 1633.12   293.4 1633.04     300 1633.66   303.2 1636.52
   309.7 1646.92     313 1650.02   335.8 1663.02   342.3 1667.63   352.1 1676.58
   355.4 1678.92  358.291679.778   371.7 1680.97     388 1681.02   391.2 1682.99
  393.291685.257   404.3 1699.35   407.6 1701.88   440.2 1720.76     463 1731.17
#Mann= 5 ,-1 , 0
       0     .12       0   281.6    .045       0     300     .12       0
  358.29    .016       0  393.29     .12       0
Bank Sta=281.6,300
XS Rating Curve= 0 ,0
Exp/Cntr=0.3,0.1

Type RM Length L Ch R = 1 ,9927.9  ,520.5,510.8,501.2
XS GIS Cut Line= 2
     2013753.038      274421.314     2013737.847      274846.661
#Sta/Elev= 30
       0 1671.66    45.8 1659.62    85.1 1648.38    91.7 1645.87   117.9 1632.68
     131 1631.18  166.481631.457  167.781631.467   180.1 1631.77   206.3 1628.89
   219.4 1628.12   231.9 1629.13   242.3 1631.26   245.6 1633.07   255.4 1641.38
   261.9  1644.6   281.6 1648.97   324.1 1660.26     334 1666.56   340.5 1672.19
   343.11673.703     347 1675.28  359.781676.656   379.8 1676.14   383.1 1677.72
  389.331684.331   396.2 1692.46   399.4 1694.75   415.8 1704.41   425.6 1709.22
#Mann= 8 ,-1 , 0
       0     .12       0  166.48     .06       0  167.78     .12       0
   206.3    .045       0   231.9     .12       0   343.1    .016       0
  359.78     .08       0  389.33     .12       0
Bank Sta=206.3,231.9
XS Rating Curve= 0 ,0
Exp/Cntr=0.3,0.1

Type RM Length L Ch R = 1 ,9417.2  ,352.5,360.6,367.7
XS GIS Cut Line= 3
     2013303.819      274447.356     2013282.118      274586.245
     2013418.837      274907.425
#Sta/Elev= 30
       0 1682.28   79.361655.466   101.3 1648.56   111.2 1643.51     121 1641.97
   137.3 1637.59  151.021635.489   186.2 1632.12   189.5 1631.24   199.3 1625.47
   209.1 1621.74     223 1619.69   248.2 1619.22   254.8 1619.48     258 1620.54
   267.8 1623.65   280.8 1625.26   287.4    1628   300.4 1638.23     320 1656.18
   339.6 1669.44  350.371677.857   355.9 1681.21   362.4  1682.3   385.2 1681.27
   388.5 1682.39  399.571691.065   408.1 1697.48     444 1711.67   489.6 1732.15
#Mann= 7 ,-1 , 0
       0     .12       0   79.36    .016       0  151.02     .12       0
     223    .045       0     258     .12       0  350.37    .016       0
  399.57     .12       0
Bank Sta=223,258
XS Rating Curve= 0 ,0
Exp/Cntr=0.3,0.1

Type RM Length L Ch R = 1 ,9056.6  ,255.3,255,254.5
XS GIS Cut Line= 3
     2012986.979      274562.373      2013004.34      274881.383
     2013071.614      275031.123
#Sta/Elev= 30
       0 1673.03    45.6 1658.53   110.8 1645.13   143.4 1629.72   153.2 1626.01
   200.11620.943  234.721617.259     251 1616.27   260.8 1616.88   263.7 1615.95
   270.6 1614.51   283.6 1615.65   293.4 1620.43   296.7 1623.88   299.9 1630.42
   303.2 1635.45   306.4 1638.03   316.2 1641.37   338.8  1661.6   361.3 1673.81
  369.861680.121   374.2 1682.29   380.6  1683.4   403.2 1683.92  408.751687.072
     416 1689.81   432.1 1693.18   451.4 1700.16   470.8 1708.64   483.6 1716.45
#Mann= 7 ,-1 , 0
       0     .12       0   200.1    .016       0  234.72     .12       0
   263.7    .045       0   283.6     .12       0  369.86    .016       0
  408.75     .12       0
Bank Sta=263.7,283.6
XS Rating Curve= 0 ,0
Exp/Cntr=0.3,0.1

Type RM Length L Ch R = 1 ,8801.6  ,65.2,65.2,65.2
XS GIS Cut Line= 3
     2012730.903      274603.606     2012754.774      274942.147
     2012824.219      275100.568
#Sta/Elev= 30
       0 1666.12   101.2 1638.11  127.821626.816  138.05 1623.01  177.681616.074
   202.3  1616.3   212.1 1615.58   215.4 1614.16   221.9 1609.02   225.2 1608.29
   231.7 1608.06     248 1608.25   254.5 1609.52   261.1 1613.27   274.1 1615.77
   303.5 1616.84   313.3 1618.42   323.1  1622.6   352.4  1637.8   417.7 1665.56
   427.5  1670.8  433.881675.383   440.6 1679.33   443.8 1679.98   466.7  1679.6
  469.11 1681.43   473.2 1685.22   479.7 1693.46  485.781697.649   512.4 1711.04
#Mann= 9 ,-1 , 0
       0     .06       0  127.82     .12       0  138.05     .06       0
  177.68    .016       0   225.2    .045       0     248     .12       0
  433.88    .016       0  469.11     .08       0  485.78     .12       0
Bank Sta=225.2,248
XS Rating Curve= 0 ,0
Exp/Cntr=0.3,0.1

Type RM Length L Ch R = 1 ,8736.3  ,128.2,123.1,117.5
XS GIS Cut Line= 3
     2012665.798      274605.776      2012689.67      274944.318
     2012759.114      275102.738
#Sta/Elev= 30
       0 1669.53   104.4 1642.28  116.281636.277     124 1631.78   143.6 1623.77
   159.9 1622.11   176.2 1615.58   182.7 1614.48  203.94 1614.79   215.4 1614.36
   228.4 1608.79   231.7 1608.32   254.5 1608.56   261.1 1609.94   270.8 1615.14
  274.641616.172  300.751616.122   319.8 1616.38   329.6 1617.75   381.8 1634.52
   417.7 1648.22   440.6 1658.97  457.931669.011   466.7 1676.07   469.9 1677.63
  484.131677.805   489.5 1677.15   492.8  1677.8   505.8 1692.37   512.4 1697.19
#Mann= 9 ,-1 , 0
       0     .06       0  116.28    .016       0  203.94     .12       0
   228.4    .045       0   254.5     .12       0  274.64    .016       0
  300.75     .12       0  457.93    .016       0  484.13     .08       0
Bank Sta=228.4,254.5
XS Rating Curve= 0 ,0
Exp/Cntr=0.3,0.1

Type RM Length L Ch R = 1 ,8613.2  ,308.7,299.7,290.1
XS GIS Cut Line= 3
     2012506.914      274686.399     2012603.717      275000.071
     2012690.508       275136.92
#Sta/Elev= 30
       0 1660.43    35.8 1653.77   81.111642.176    97.5 1637.76   110.5 1637.16
   113.8 1635.16  121.291627.305   136.5  1612.5   139.8 1611.18   162.5 1608.42
   176.2 1608.26   185.3 1607.92   198.3 1608.45   211.3 1614.54  219.991614.637
  253.961614.969   282.8 1614.11   354.2 1624.55   370.4 1628.75   386.6 1634.69
   402.8 1642.38  431.781658.918   451.4 1672.52   461.2 1672.83   470.9 1671.74
   474.1 1672.82  477.971676.628   483.8 1685.63   487.1 1689.42   490.3 1691.65
#Mann= 9 ,-1 , 0
       0     .06       0   81.11    .016       0  121.29     .12       0
   176.2    .045       0   198.3     .12       0  219.99    .016       0
  253.96     .12       0  431.78    .016       0  477.97     .12       0
Bank Sta=176.2,198.3
XS Rating Curve= 0 ,0
Exp/Cntr=0.3,0.1

Type RM Length L Ch R = 1 ,8313.5  ,370.2,353,335.6
XS GIS Cut Line= 2
      2012227.43      274892.234     2012520.399      275226.436
#Sta/Elev= 30
       0 1657.76    22.9 1654.48    29.4 1650.91    42.5 1639.24    55.6 1626.39
    68.6 1610.53    75.2 1604.18    78.4 1601.95    81.7 1601.04      85 1600.94
   101.3 1601.46   111.1 1602.64   124.2 1605.78  152.49 1604.65   160.1 1605.39
   169.9 1608.94   173.2  1609.6   189.5 1611.18  205.841611.639     232 1612.42
   290.8 1615.79   339.9 1620.38  372.331625.594   388.9 1629.28   411.8 1637.16
   421.6 1641.76   428.1 1646.15  434.76 1651.58   441.2 1657.57   444.4 1659.82
#Mann= 7 ,-1 , 0
       0     .12       0    78.4    .045       0   101.3     .12       0
  152.49    .016       0  205.84     .06       0  372.33     .12       0
  434.76    .016       0
Bank Sta=78.4,101.3
XS Rating Curve= 0 ,0
Exp/Cntr=0.3,0.1

Type RM Length L Ch R = 1 ,7960.4  ,493.5,512.2,530
XS GIS Cut Line= 3
     2011949.623      275131.712     2012038.164      275242.389
     2012365.885      275272.008
#Sta/Elev= 30
       0 1649.56    12.9 1648.13    35.4 1644.35    48.3 1642.95    67.6  1639.6
    83.8 1635.89    99.9 1630.02   122.4  1618.9   135.3 1611.61   141.7 1608.73
     158 1604.21   167.8  1597.9   171.1 1596.37   184.4 1595.43   190.6 1595.36
   203.6 1595.51   210.2 1598.62   213.4 1599.55     233 1599.72   236.2 1600.09
   242.7 1602.25     246 1602.68  261.081602.241   337.2 1602.98   365.61604.931
  379.031607.737   405.6 1617.06   431.7 1621.01  458.141626.828   470.8 1629.87
#Mann= 7 ,-1 , 0
       0     .12       0   184.4    .045       0   203.6    .016       0
  261.08     .06       0   365.6     .12       0  379.03     .06       0
  458.14     .12       0
Bank Sta=184.4,203.6
XS Rating Curve= 0 ,0
Exp/Cntr=0.3,0.1

Type RM Length L Ch R = 1 ,7448.2  ,416,417.4,418
XS GIS Cut Line= 2
     2011652.748      275450.722     2011971.354      275847.095
#Sta/Elev= 30
       0 1616.38    22.8 1613.16    52.2 1611.38    71.7 1608.65    78.2 1606.63
    94.5  1595.2   104.3 1592.23  141.94  1591.9   211.9 1591.89   244.5 1591.94
   254.3 1590.43     264 1585.94   274.5 1584.83   289.5 1584.73   293.4 1584.86
   299.9 1586.38  304.881589.567   309.7 1594.38   319.5 1606.04   322.7 1609.07
     326 1610.86   345.6  1612.8   358.6 1612.28   361.8 1612.89  367.33 1617.56
   374.9 1627.92   387.9 1640.96   391.2 1643.53   446.6 1681.53   508.6 1719.83
#Mann= 7 ,-1 , 0
       0     .12       0  141.94     .06       0   211.9     .12       0
   274.5    .045       0   293.4     .12       0  304.88    .016       0
  367.33     .12       0
Bank Sta=274.5,293.4
XS Rating Curve= 0 ,0
Exp/Cntr=0.3,0.1

Type RM Length L Ch R = 1 ,7030.9  ,284.6,284.6,284.7
XS GIS Cut Line= 2
     2011295.139      275635.724     2011605.469      276061.071
#Sta/Elev= 30
       0 1606.37     6.5 1602.48    13.1 1600.96    32.7 1600.32   65.111597.345
  132.791591.233   166.8 1589.15   170.1 1588.34   183.1 1581.35   189.7 1579.91
   212.6 1579.01   222.4  1580.4   245.3 1579.44   264.9 1580.31     314 1578.09
     327 1576.74   336.8 1577.41   343.4 1581.11   349.9  1587.4  359.27 1590.99
   369.6 1597.16   389.2 1596.99   392.4 1598.04  401.031604.581   408.8  1613.5
   418.6 1621.28   467.7 1654.67   490.6 1669.19   503.6 1679.96   526.5  1693.8
#Mann= 7 ,-1 , 0
       0     .12       0   65.11     .06       0  132.79     .12       0
     314    .045       0   336.8     .12       0  359.27    .016       0
  401.03     .12       0
#XS Ineff= 2 , 0
          204.55 1593.89
Permanent Ineff=
       F       F
Bank Sta=314,336.8
XS Rating Curve= 0 ,0
Exp/Cntr=0.3,0.1

Type RM Length L Ch R = 1 ,6746.2  ,253.5,265.5,276.8
XS GIS Cut Line= 2
     2011078.993      275821.922     2011389.323      276247.269
#Sta/Elev= 30
       0 1583.65     6.5 1581.85   26.321581.177    81.8 1580.22   143.9 1577.55
  235.49 1577.35   261.6 1577.13     278 1573.48   284.5 1570.79   287.8 1570.33
   304.1 1569.53     314 1570.56   333.6 1575.24   343.4 1586.92   346.6 1589.12
  354.871591.793   359.7 1594.81   366.3 1600.27   369.6 1601.47  386.041601.589
   392.4 1602.05   395.7 1604.39   402.2 1614.74   405.5 1618.12   415.3 1625.19
     448 1645.58   461.1 1651.77     484 1660.27   516.7 1670.46   526.5 1672.69
#Mann= 7 ,-1 , 0
       0     .12       0   26.32     .06       0  235.49     .12       0
   287.8    .045       0     314     .12       0  354.87    .016       0
  386.04     .12       0
Bank Sta=287.8,314
XS Rating Curve= 0 ,0
Exp/Cntr=0.3,0.1

Type RM Length L Ch R = 1 ,6480.8  ,590.6,574.8,557.1
XS GIS Cut Line= 3
     2011005.612      275832.667     2011016.463      276006.278
     2011075.087      276500.307
#Sta/Elev= 30
       0 1601.09    19.3 1587.34      29 1581.57    35.4 1579.26   97.121575.981
   239.4 1575.02   278.7 1572.47  312.411572.527   327.8 1573.07   337.6 1570.76
   350.7  1570.6   360.9 1568.07   370.3  1567.3   386.7 1568.39     390 1570.77
   399.8 1585.33   403.1  1589.1  411.691593.501   439.1 1594.18  456.891598.521
  486.641605.732  533.79 1609.89   560.2 1612.78  585.641617.828   596.2 1621.04
   615.8 1621.68   620.3 1624.54   628.9 1631.15   658.4 1639.53   671.4  1644.7
#Mann= 11 ,-1 , 0
       0     .12       0   97.12     .06       0  312.41     .12       0
   360.9    .045       0   386.7     .12       0  411.69    .016       0
  456.89     .06       0  486.64     .08       0  533.79     .12       0
  585.64    .016       0   620.3     .12       0
Bank Sta=360.9,386.7
XS Rating Curve= 0 ,0
Exp/Cntr=0.3,0.1

Type RM Length L Ch R = 1 ,5906    ,523.6,525.9,528
XS GIS Cut Line= 2
     2010358.941       276077.13     2010851.562      276515.498
#Sta/Elev= 30
       0 1661.56    19.7 1655.42    39.4 1648.11    75.5 1631.21    91.9 1622.76
   101.7 1618.48   134.5 1597.51   137.8 1592.77   154.2 1564.46   157.5 1561.73
   160.8 1561.38   170.6 1560.81   179.2 1561.59     187 1562.21   193.6  1564.2
   196.8 1564.51   229.6  1566.2   255.9 1565.21   288.7 1565.73   337.9 1563.95
   354.3 1569.28  373.241570.279   423.2 1570.21   462.6 1571.15     502 1573.01
     561 1576.96   600.4 1582.97  627.61 1591.64   652.9 1602.13   659.4  1606.8
#Mann= 5 ,-1 , 0
       0     .12       0   160.8    .045       0   179.2     .12       0
  373.24     .06       0  627.61     .12       0
Bank Sta=160.8,179.2
XS Rating Curve= 0 ,0
Exp/Cntr=0.3,0.1

Type RM Length L Ch R = 1 ,5380.1  ,358.2,363.2,367.8
XS GIS Cut Line= 4
     2010011.719      276357.078     2010102.864      276537.199
     2010254.774      276693.449      2010506.51      276741.193
#Sta/Elev= 30
       0 1697.21      26 1678.31    55.4 1661.42    74.9  1648.7    94.4 1634.97
   110.7 1624.63   133.5 1608.61     166 1591.14   185.6 1582.06   205.1 1571.34
   231.1 1559.15   237.6  1557.7   244.2 1557.15   263.7 1556.95   270.2 1557.49
   279.9 1554.06   299.4 1553.52   307.1 1554.16     319 1556.51   341.7  1556.8
  359.541559.136   403.5 1559.64   491.2 1562.14   546.3  1565.6  594.981570.289
   624.1    1573   640.3 1578.28   656.6 1582.19  664.141584.816     676 1590.18
#Mann= 6 ,-1 , 0
       0     .12       0   279.9    .045       0   307.1     .12       0
  359.54     .06       0  594.98     .12       0  664.14    .016       0
Bank Sta=279.9,307.1
XS Rating Curve= 0 ,0
Exp/Cntr=0.3,0.1

Type RM Length L Ch R = 1 ,5017    ,404,405.1,406.1
XS GIS Cut Line= 2
     2009802.615      276598.923     2010099.294      277100.476
#Sta/Elev= 30
       0 1610.86    42.6 1593.23   101.5 1564.08   114.6 1559.27   134.2 1553.89
   151.11552.272   248.8 1550.81  289.921552.182  324.24 1551.93     347  1552.2
   356.8 1549.02   363.4 1547.99   379.8 1547.08   386.3  1547.8   392.8 1549.95
     406 1559.02   412.5 1567.39     419 1574.37  425.571579.203   432.1 1580.03
   451.8 1578.89   458.3 1581.43  464.131585.363   471.4 1589.61   474.7 1589.95
   500.9 1598.45   527.1 1608.42   559.8 1624.26   572.9 1629.58   582.7 1635.13
#Mann= 8 ,-1 , 0
       0     .12       0   151.1     .06       0  289.92     .08       0
  324.24     .12       0   363.4    .045       0   386.3     .12       0
  425.57    .016       0  464.13     .12       0
Bank Sta=363.4,386.3
XS Rating Curve= 0 ,0
Exp/Cntr=0.3,0.1

Type RM Length L Ch R = 1 ,4611.8  ,379.9,380.2,380.3
XS GIS Cut Line= 3
     2009495.226      276769.404     2009510.417      276869.231
     2009740.451      277303.258
#Sta/Elev= 30
       0 1625.02    52.1 1584.76    78.2 1568.12      88 1564.28   107.5  1550.8
   123.9 1546.56  144.311545.686  177.741544.172   244.61544.267   294.2 1547.06
     304 1546.13   313.8 1542.34   320.4 1541.26   326.9 1541.02   340.7 1541.52
   356.4 1543.41   366.2 1543.38   382.6  1545.9   408.8 1561.79  418.061570.016
   425.2 1573.68  458.091575.099   467.8 1576.14   477.6 1584.74   484.1 1588.73
   497.2 1591.08   510.3 1591.82   533.2 1597.85   562.7 1607.89   592.2 1620.79
#Mann= 8 ,-1 , 0
       0     .12       0  144.31     .08       0  177.74     .06       0
   244.6     .12       0   320.4    .045       0   340.7     .12       0
  418.06    .016       0  458.09     .12       0
Bank Sta=320.4,340.7
XS Rating Curve= 0 ,0
Exp/Cntr=0.3,0.1

Type RM Length L Ch R = 1 ,4231.7  ,245.1,262.4,278.6
XS GIS Cut Line= 2
     2009189.236      277064.543     2009427.951      277520.272
#Sta/Elev= 30
       0 1547.61    75.4 1543.71  103.551543.195  189.531539.521  221.081537.944
   245.2 1534.75   258.9 1534.66   262.2  1534.8     272 1537.26   288.4 1538.28
   291.6 1539.23  297.881543.196   301.5    1545     308 1546.29   324.4 1546.68
     331  1545.8   334.2 1547.74   340.8 1555.28   344.1 1560.41   347.4 1567.16
   353.9 1583.06   357.2 1587.07  374.721596.806   399.8 1611.18     403 1612.35
   416.2 1613.21   419.4 1615.31   429.3 1625.36   452.2  1636.7   514.5 1661.86
#Mann= 8 ,-1 , 0
       0     .08       0  103.55     .06       0  189.53     .08       0
  221.08     .12       0   245.2    .045       0   262.2     .12       0
  297.88    .016       0  374.72     .12       0
Bank Sta=245.2,262.2
XS Rating Curve= 0 ,0
Exp/Cntr=0.3,0.1

Type RM Length L Ch R = 1 ,3969.2  ,93.8,94,93.9
XS GIS Cut Line= 3
     2008991.753      277066.713     2009124.132      277270.706
     2009026.476       277637.46
#Sta/Elev= 30
       0 1550.08    8.611549.561    25.9 1549.09    61.6 1544.66   72.181545.277
   94.441543.203  127.131542.113  162.341542.008  171.391541.395  197.561540.157
   247.61537.663   269.4 1536.02   308.6 1536.96   318.4 1538.06  348.071535.969
     374 1533.78   384.2 1530.66   390.4 1529.52   406.8 1530.65   416.6 1536.38
   423.1  1538.6  454.311538.909   521.3 1540.14   531.1 1536.25   534.4 1535.88
   540.9 1536.71  544.321538.757   550.7 1541.79     590 1544.99   622.7 1543.73
#Mann= 14 ,-1 , 0
       0     .06       0    8.61    .016       0   72.18     .08       0
   94.44    .016       0  127.13     .06       0  162.34     .08       0
  171.39     .12       0  197.56    .016       0   247.6     .06       0
  348.07     .12       0   384.2    .045       0   406.8    .016       0
  454.31     .08       0  544.32     .12       0
#XS Ineff= 2 , 0
                          465.34         1541.66
Permanent Ineff=
       F       F
Bank Sta=384.2,406.8
XS Rating Curve= 0 ,0
Exp/Cntr=0.3,0.1

Type RM Length L Ch R = 1 ,3875.2  ,161.1,151.9,143.1
XS GIS Cut Line= 3
     2008898.437      277062.373     2009030.816      277266.366
      2008933.16       277633.12
#Sta/Elev= 30
       0 1591.74    71.3 1559.53    90.8 1551.91   98.061550.722   132.31546.853
   152.4 1546.01  167.521543.425     201 1540.79  234.291540.525  237.941540.275
  299.771536.798  330.331535.521   364.2    1535   377.3 1528.73   387.1 1527.94
   398.8 1528.41   416.6 1530.99   426.4 1535.93   429.7 1536.58   442.8 1536.57
   452.6 1533.89  464.981535.528   472.2 1537.47  499.031537.841   537.6 1540.18
   562.2 1539.06   599.8 1540.72   606.4 1542.14  614.72 1546.02   622.7 1549.97
#Mann= 14 ,-1 , 0
       0     .12       0   98.06     .08       0   132.3    .016       0
  167.52     .08       0  234.29    .016       0  237.94     .12       0
  299.77     .08       0  330.33     .06       0   377.3    .045       0
   398.8     .12       0  464.98    .016       0  499.03     .08       0
   562.2     .06       0  614.72     .12       0
#XS Ineff= 2 , 0
                          431.53         1544.76
Permanent Ineff=
       F       F
Bank Sta=377.3,398.8
XS Rating Curve= 0 ,0
Exp/Cntr=0.3,0.1

Type RM Length L Ch R = 1 ,3723.3  ,292.2,293.7,293.6
XS GIS Cut Line= 3
     2008755.208      277214.283     2008828.993      277309.769
     2008885.417      277743.797
#Sta/Elev= 30
       0  1621.2    35.9 1595.33    52.2 1581.85    65.2 1572.65      75 1562.78
    88.1  1553.7   101.1 1546.16   117.4  1539.6     137 1533.77   150.1 1532.01
  167.59 1532.04  202.571533.007   231.7 1532.48   244.8 1527.76     255 1526.56
   264.4  1526.5     270  1526.7   277.4 1527.67   287.2 1532.38  301.881533.742
  339.51 1535.17  356.011535.774  393.411536.766  429.911539.225   447.3 1544.22
   460.4 1550.75   476.7 1560.61   532.2 1597.36   545.3 1609.91   558.4 1618.77
#Mann= 10 ,-1 , 0
       0     .12       0  167.59     .06       0  202.57     .12       0
     255    .045       0     270     .12       0  301.88    .016       0
  339.51     .08       0  356.01     .06       0  393.41     .08       0
  429.91     .12       0
Bank Sta=255,270
XS Rating Curve= 0 ,0
Exp/Cntr=0.3,0.1
